--- GLADYFK.prj (project) ---

Proj Title=GLADYFK
Current Plan=p01
Default Exp/Contr=0,0
English Units
Geom File=g01
Flow File=f01
Plan File=p01
BEGIN DESCRIPTION:
---------- MODELED AS PART OF WVEMD CTP PROGRAM, 2023----------
Stream Name: Glady Fork
Flood Zone:  AFH
Upshur County, WV
HEC-RAS Version: RAS 6.3
Vertical Datum: NAVD88
Projection: NAD 1983 StatePlane West Virginia S FIPS 4702 (US Feet)
Terrain: 1-meter LIDAR (FEMA Region III 3DEP collected 2016-2018)
Land Use: 2019 NLCD
Hydrologic Method:
WV 2010 Regional Regression Equations
Additional Model Notes:
None
END DESCRIPTION:
DSS Export Rating Curves= 0
DSS Export Rating Curve Sorted= 0
DSS Export Volume Flow Curves= 0
DXF OffsetX= 0
DXF OffsetY= 0
DXF ScaleX= 0
DXF ScaleY= 0

--- GLADYFK.p01 (plan) ---

Plan Title=Floodplain
Program Version=4.00
Geom File=g01
Flow File=f01
K Sum by GR=0
Std Step Tol=0.01
Critical Tol=0.01
Num of Std Step Trials=20
Max Error Tol=0.3
Flow Tol Ratio=0.001
Split Flow NTrial=30
Split Flow Tol=0.02
Split Flow Ratio=0.02
Log Output Level=0
Friction Slope Method=1
Unsteady Friction Slope Method=2
Unsteady Bridges Friction Slope Method=1
Global Log Level=0
CheckData=False
Run HTab=0
Run UNet=0
Run PostProcess=0
UNET Theta=0
UNET Theta Warmup=0
UNET ZTol=0
UNET ZSATol=0
UNET MxIter=0
UNET MaxInSteps=0
UNET DtIC=0
UNET DtMin=0
UNET MaxCRTS=0
UNET WFStab=0
UNET SFStab=0
UNET WFX=0
UNET SFX=0
UNET DSS MLevel=0
UNET DZMax Abort=0
UNET Convert EG Bridges=0
UNET Use Existing IB Tables=0
UNET Froude Limit=0
UNET Froude Power=0
Write IC File=0
Echo Input=False
Echo Output=False
Write Detailed=0

--- GLADYFK.f01 (steady flow) ---

Flow Title=Flows
Program Version=6.31
Number of Profiles= 1
Profile Names=01pct
River Rch & RM=GLADYFK,Main            ,10122
     977
River Rch & RM=GLADYFK,Main            ,5031
    1180
River Rch & RM=GLADYFK,Main            ,470
    1370
River Rch & RM=GLADYFK,Main            ,0
    2150
Boundary for River Rch & Prof#=GLADYFK,Main            , 1
Up Type= 0
Dn Type= 1
Dn Known WS=1250.44
DSS Import GetInterval= 0
DSS Import GetPeak= 0
DSS Import FillOption= 0

--- GLADYFK.g01 (geometry) ---

Geom Title=Geometry
Program Version=6.31

River Reach=GLADYFK         ,Main
Reach XY= 30
2169342.34100001711955.4070000052169414.31100002712041.457000017
2169653.37300003711967.7690000092170049.05100003712128.536000013
2170161.19900002712214.2710000132170180.22900003712370.001000002
2170320.50600001712437.6220000092170665.04800002712286.985000014
2170698.87200002712350.142000005     2170958.108712335.174999997
     2170971.529712471.8760000172171210.64800002712622.942000002
2171513.12299998713323.327999994     2171857.979713377.613000005
2172041.52500001713652.4730000052172065.41899998713989.688999996
2171915.29800002714247.9229999932172028.76200002714423.199000001
2172062.41500004714743.788000003     2171869.111 715530.51000002
     2172090.745715889.8460000162172265.01900001716402.422000021
2172026.18600003716807.8589999972172187.86900002717150.083000019
      2172099.73717459.1969999972172225.32799999718008.231000021
2172075.17800002      718352.772     2171810.447718614.069000006
2171688.28400004718662.5450000022171389.82671208718570.855522095

Type RM Length L Ch R = 1 ,10122   ,262.1,262.1,262.1
XS GIS Cut Line= 2
2169163.12460855 712091.352683732169378.76496317711931.913974117
#Sta/Elev= 30
       0  1448.8     6.3 1448.05    10.4 1446.67    16.6 1441.39    19.5 1440.39
    21.2 1440.22    37.3 1440.67    41.1 1440.38    48.1 1438.93    50.8 1438.73
    56.6 1439.54    59.5 1439.52    77.7 1436.85    97.9 1435.48   130.6 1434.69
   159.6 1434.95   165.3 1435.49   170.4 1435.46     192 1432.99   205.5 1432.12
   215.2 1432.06     219 1431.19   225.2 1430.14  230.92 1431.19   235.1 1432.11
   240.1 1432.65     254 1437.79   256.8 1439.57   265.4 1446.49   268.2 1448.15
#Mann= 5 ,-1,0
       0      .1       0      50     .06       0     210      .1       0
     219    .045       0  230.92      .1       0
Bank Sta=219,230.92
XS Rating Curve= 0 ,0
Exp/Cntr(USF)=0,0
Exp/Cntr=0.3,0.1

Type RM Length L Ch R = 1 ,9860    ,273.8,279.9,285.4
XS GIS Cut Line= 3
2169523.04460733712239.9138608472169561.50392696712083.262485734
2169528.67280044711926.611110622
#Sta/Elev= 30
       0 1452.17     6.9  1451.2    19.7 1447.26    52.2 1440.42    68.7 1438.51
    92.5 1437.42   122.2 1438.56   171.6 1439.34   179.8 1439.06     188 1439.43
     192 1438.62     198 1435.94   204.7 1433.99   214.9 1433.08   228.8    1431
   245.2 1430.31   248.71429.012   253.3 1428.02   257.4 1427.94   261.5 1428.31
   263.81429.026   269.7 1430.25   273.8 1430.55     282 1429.52     286 1429.41
   290.1  1430.3   298.3 1432.92   302.4 1434.94   310.6 1441.17   321.4 1451.29
#Mann= 5 ,-1,0
       0     .06       0      80     .05       0   181.3      .1       0
   248.7    .045       0   263.8      .1       0
Bank Sta=248.7,263.8
XS Rating Curve= 0 ,0
Exp/Cntr(USF)=0,0
Exp/Cntr=0.3,0.1

Type RM Length L Ch R = 1 ,9580    ,244,244.4,244.6
XS GIS Cut Line= 2
2169716.31861189712300.6937142612169803.27419556711999.303972803
#Sta/Elev= 30
       0 1453.51     7.8    1450      12 1448.97    16.1 1448.38    49.5 1440.94
      58  1439.4    70.3 1437.64    86.9 1436.31    95.2 1435.91   111.9 1435.81
   124.4 1436.12     141 1435.94   149.4 1435.76   178.5 1434.22     216 1431.56
   228.9 1430.88   236.8 1430.76     241 1429.84  246.161427.416   249.3 1426.37
   257.6 1426.03  263.391427.358   274.3 1430.94   278.4 1433.06   282.6    1436
     287 1438.29   290.9 1439.29   299.2 1443.09   307.6 1445.57   313.7 1447.87
#Mann= 5 ,-1,0
       0     .05       0      40     .06       0     150     .05       0
  246.16    .045       0  263.39      .1       0
Bank Sta=246.16,263.39
XS Rating Curve= 0 ,0
Exp/Cntr(USF)=0,0
Exp/Cntr=0.3,0.1

Type RM Length L Ch R = 1 ,9335    ,244.4,256.6,266.6
BEGIN DESCRIPTION:
Structure1 XS4
END DESCRIPTION:
XS GIS Cut Line= 3
2169940.49189874712343.1897170572170000.07865504712189.476784479
2170040.92580661712061.411654683
#Sta/Elev= 30
       0 1444.27    10.7 1441.15    27.9 1435.69    36.5 1433.23    41.5  1432.1
    47.7 1430.99    57.9 1429.85    66.2 1429.27      88 1428.43    97.1 1428.41
   106.4 1428.75   130.9  1428.4   143.7 1428.46   186.2 1427.78     203 1427.06
   228.1  1426.4   232.3 1425.74  234.081425.206   236.5 1424.47   240.7 1424.12
   244.9 1424.43  250.791425.195   261.7 1427.41   265.9 1429.47     270 1433.07
   276.1 1439.24   279.8 1442.44   286.1 1446.83   295.3 1452.01   299.3 1454.79
#Mann= 5 ,-1,0
       0     .06       0      90     .05       0  234.08    .045       0
  250.79     .05       0  294.86      .1       0
#XS Ineff= 2 , 0
          221.01 1429.68
Permanent Ineff=
       F       F
Bank Sta=234.08,250.79
XS Rating Curve= 0 ,0
Exp/Cntr(USF)=0,0
Exp/Cntr=0.3,0.1

Type RM Length L Ch R = 1 ,9079    ,40.4,40,39.6
XS GIS Cut Line= 4
2170057.69548201712429.7545521052170107.99371203712304.373456986
2170280.75719775712235.122270729 2170288.0467963712124.320372718
#Sta/Elev= 30
       0 1448.29     5.4  1446.9    17.4 1436.56    22.2 1433.95    35.1 1428.76
    49.6 1425.44    65.3 1424.02    91.1 1424.52   112.7 1424.16   129.9  1424.8
   148.2  1424.6   153.1 1424.07   162.61419.738   169.8 1417.88  181.761419.741
   199.9 1427.77   204.2 1428.85   212.9 1429.88   261.9 1433.76   286.1 1434.19
   307.7 1433.14   321.2 1433.53   339.2 1434.97   352.6 1436.87   371.3 1438.47
   379.3 1439.72   395.3 1443.51   407.3 1447.35   422.6 1453.28   432.3 1455.91
#Mann= 7 ,-1,0
       0     .06       0      80     .05       0  145.09      .1       0
   162.6    .045       0  181.76      .1       0  245.09     .05       0
  255.09      .1       0
Bank Sta=162.6,181.76
XS Rating Curve= 0 ,0
Exp/Cntr(USF)=0,0
Exp/Cntr=0.3,0.1

Type RM Length L Ch R = 1 ,9039    ,24.5,24.6,24.7
BEGIN DESCRIPTION:
Structure1 XS3
END DESCRIPTION:
XS GIS Cut Line= 4
2170091.50669036712444.4117351712170113.82239165712346.463605578
2170293.18361042712268.0616841462170302.56393228712135.799145877
#Sta/Elev= 30
       0 1446.94     3.3 1446.75     7.4 1445.79    11.5 1443.23    19.7 1436.96
    23.8 1434.93    36.1 1430.04    44.3 1427.54    48.4 1426.66    60.8 1424.46
    73.1 1423.44   100.5 1423.76   130.6 1422.74   133.6 1422.47   136.6 1421.64
  142.651418.762   146.7  1417.5     151 1417.09  155.661418.779   159.8 1421.04
   164.1 1422.18   181.6 1424.94   264.5 1428.59   307.1 1431.06     322 1432.53
   339.1 1435.06   369.1 1438.45   399.1    1441   411.4 1443.69   428.8 1450.69
#Mann= 5 ,-1,0
       0     .06       0      90     .05       0  110.46      .1       0
  142.65    .045       0  155.66      .1       0
Bank Sta=142.65,155.66
XS Rating Curve= 0 ,0
Exp/Cntr(USF)=0,0
Exp/Cntr=0.3,0.1

Type RM Length L Ch R = 1 ,9014    ,56.7,49,40.5
BEGIN DESCRIPTION:
Structure1 XS2
END DESCRIPTION:
XS GIS Cut Line= 4
2170106.17135089712466.5806531832170128.48705218712366.416929088
2170307.84827094712290.2306021582170317.22859281 712157.96806389
#Sta/Elev= 30
       0 1446.63    13.7 1446.47    21.9 1445.74      26 1444.12    34.2  1438.4
    38.3  1436.2    54.7 1429.96      67 1426.33    79.3 1424.73    91.6 1423.87
   119.7 1423.36   132.7 1421.31   139.9 1417.59   141.4  1416.6   145.7 1415.39
   149.1 1416.25  151.711417.594   158.2  1421.4   163.1 1422.74   167.5  1423.2
   179.6 1422.88   271.1 1424.97   289.2 1423.91   297.5 1424.08   315.5 1428.74
   324.2 1430.52   350.1 1432.46   406.8 1440.63   418.8 1441.65   430.1 1441.98
#Mann= 5 ,-1,0
       0     .05       0      10     .06       0  122.62      .1       0
   139.9    .045       0  151.71      .1       0
Bank Sta=139.9,151.71
XS Rating Curve= 0 ,0
Exp/Cntr(USF)=0,0
Exp/Cntr=0.3,0.1

Type RM Length L Ch R = 1 ,8965    ,337.8,333.4,325.3
XS GIS Cut Line= 4
2170156.83402234712477.1369427022170223.67074776712332.050823462
2170324.58583615712287.5716612812170336.39498581712164.231653757
#Sta/Elev= 30
       0 1446.21    13.2 1446.13    17.6 1445.41    26.4 1441.53    35.2 1439.32
    48.4  1433.9    62.8  1432.7    65.8 1431.63    68.8 1429.75    79.2 1421.99
    83.6 1419.16    93.21415.726   101.2 1415.12  105.271415.733   110.1 1416.57
   118.9 1416.27   132.1 1417.16   159.7  1421.7     204 1421.81   225.9 1423.51
   247.3 1422.39     270 1423.29   284.5 1426.16   304.2 1431.11   312.6 1431.91
   324.7 1432.35   336.7 1433.52   352.8 1435.79   375.3 1440.08   393.9 1443.12
#Mann= 5 ,-1,0
       0     .05       0      20     .06       0    93.2    .045       0
  105.27     .06       0     130      .1       0
Bank Sta=93.2,105.27
XS Rating Curve= 0 ,0
Exp/Cntr(USF)=0,0
Exp/Cntr=0.3,0.1

Type RM Length L Ch R = 1 ,8632    ,301.2,305.9,307.1
BEGIN DESCRIPTION:
Structure1 XS1
END DESCRIPTION:
XS GIS Cut Line= 2
2170493.82600292712518.9263574192170465.68503733712294.736664893
#Sta/Elev= 30
       0 1437.04     9.8 1435.98    13.9 1435.41    23.2 1433.64      30 1432.08
    45.4 1427.09    54.2 1423.66    58.2  1422.3    78.5 1415.98    86.4 1413.68
    90.5 1412.62    94.5 1412.13   102.5 1412.38   130.8 1411.82   142.9 1411.04
   150.9 1411.04     159 1411.25     167 1409.98   171.4 1409.83   179.1 1409.88
   183.2  1409.1  185.611408.371   187.2 1407.89   191.2 1407.49   195.3 1407.57
   198.3 1408.38   199.3 1408.62   211.4 1415.45   219.5 1419.71   225.9 1423.66
#Mann= 4 ,-1,0
       0     .06       0     160      .1       0  185.61    .045       0
   198.3      .1       0
Bank Sta=185.61,198.3
XS Rating Curve= 0 ,0
Exp/Cntr(USF)=0,0
Exp/Cntr=0.3,0.1

Type RM Length L Ch R = 1 ,8326    ,369.9,386.2,396.6
XS GIS Cut Line= 2
2170696.31699937712512.6529365532170734.53312548712252.088440358
#Sta/Elev= 30
       0 1434.25     3.5 1432.84      17  1424.4    27.8 1418.57    43.9 1411.31
      52 1408.64    56.1 1407.82    60.1 1407.26    64.2 1407.12    68.2 1407.36
     118 1406.56   149.1  1406.5   153.1 1406.18  157.141404.352   161.2 1403.58
  164.831404.333   169.3 1405.13   181.4 1405.35   197.6 1405.55   209.7 1405.39
   221.8 1404.78   225.9 1405.21   229.9 1406.72     238 1411.21     242 1415.05
   246.2  1419.8   250.1 1423.65   258.2 1433.19   262.2 1436.17   263.4 1436.66
#Mann= 4 ,-1,0
       0     .07       0      60     .05       0  157.14    .045       0
  164.83      .1       0
#XS Ineff= 2 , 0
          101.65 1410.43
Permanent Ineff=
       F       F
Bank Sta=157.14,164.83
XS Rating Curve= 0 ,0
Exp/Cntr(USF)=0,0
Exp/Cntr=0.3,0.1

Type RM Length L Ch R = 1 ,7939    ,156,151,146.9
BEGIN DESCRIPTION:
Structure2 XS4
END DESCRIPTION:
XS GIS Cut Line= 3
2170830.08103251712555.9564396922170866.38287812712471.533542925
2171240.62178151712382.961353834
#Sta/Elev= 30
       0 1425.77     7.4 1425.45    11.7 1424.54      22 1419.23    29.1  1414.7
    40.2 1409.44    49.4  1406.5    59.6 1404.57    72.7 1403.18    90.1 1402.74
   175.1 1402.05   180.1 1401.35183.48941400.145   188.4 1399.16196.5993 1400.16
   208.8 1401.79   245.8 1401.05   258.2 1401.37   299.3 1406.94   323.9 1407.74
   333.5 1408.75   360.9 1413.28   373.3 1413.14   377.4 1413.92   385.6 1420.86
   389.7  1423.5   406.1 1427.28   414.4 1429.78   427.7  1434.9   476.5 1448.85
#Mann= 5 ,-1,0
       0     .06       0   141.9     .05       0183.4894    .045       0
196.5993     .05       0   331.9     .06       0
#XS Ineff= 2 , 0
          149.61 1406.54
Permanent Ineff=
       F       F
Bank Sta=183.4894,196.5993
XS Rating Curve= 0 ,0
Exp/Cntr(USF)=0,0
Exp/Cntr=0.3,0.1

Type RM Length L Ch R = 1 ,7789    ,80.2,69.6,67.2
XS GIS Cut Line= 2
2170944.69084525712630.7586715762171183.29471406712439.450447141
#Sta/Elev= 30
       0 1423.07     3.6 1419.04     8.9 1413.97    12.1 1411.92      15 1410.76
    21.7  1411.3    28.1 1411.32    34.9 1411.06    43.4 1410.27    60.9 1406.86
      69 1404.44    80.4  1402.6    86.5 1402.22   104.8 1401.93   117.4 1399.69
     124 1399.55   153.1 1400.11  161.361399.119   171.5 1398.68   177.2 1399.12
   183.9 1400.26   194.2 1404.29   197.1 1404.67   209.5 1405.27   235.2 1407.31
   250.6 1407.46   255.7 1408.99   260.8 1411.67   276.2 1416.72   305.8 1427.52
#Mann= 4 ,-1,0
       0     .05       0     120     .06       0  161.36    .045       0
   177.2     .06       0
Bank Sta=161.36,177.2
XS Rating Curve= 0 ,0
Exp/Cntr(USF)=0,0
Exp/Cntr=0.3,0.1

Type RM Length L Ch R = 1 ,7719    ,24,23.8,25
BEGIN DESCRIPTION:
Structure2 XS3
END DESCRIPTION:
XS GIS Cut Line= 3
2171050.65749082712663.8507076242171114.07337105712516.599396131
2171201.52493927712459.623938336
#Sta/Elev= 30
       0 1402.77    11.6 1403.81    15.4 1403.85    30.6 1403.61    50.8 1402.82
    55.2 1402.25    59.5 1400.33    63.9 1397.71    65.81396.906    68.2 1395.94
    72.6 1395.75    76.9  1395.8    79.3  1396.1    82.3  1396.9    85.7 1398.46
      90 1399.56   125.2 1402.75     131 1403.02   135.3 1403.54   172.4 1405.76
   177.2 1405.83   186.7 1405.39   191.5 1405.61   196.1 1406.55     201 1408.15
   205.8 1409.47   215.3 1411.66   224.9 1414.47   248.8 1423.15   264.7 1429.94
#Mann= 4 ,-1,0
       0     .05       0    65.8    .045       0    82.3     .05       0
     120     .06       0
Bank Sta=65.8,82.3
XS Rating Curve= 0 ,0
Exp/Cntr(USF)=0,0
Exp/Cntr=0.3,0.1

Type RM Length L Ch R = 1 ,7695    ,57.5,54.8,50.4
BEGIN DESCRIPTION:
Structure2 XS2
END DESCRIPTION:
XS GIS Cut Line= 3
2171073.37056071712674.290568097 2171129.4300071 712537.60347968
2171225.16557203 712504.17201256
#Sta/Elev= 30
       0 1403.24    18.3 1403.63    53.1 1402.71    61.3 1401.59    66.1 1399.17
    67.4 1398.04   68.561397.319    70.6  1396.1    73.5 1395.82      79 1395.73
    83.3 1396.1285.831861397.315    87.7 1398.18    91.9 1400.76    96.3 1402.04
   100.6 1402.38   112.8 1402.74   119.5 1403.24   123.3 1403.16   144.4 1403.82
   154.9 1404.72   167.6 1405.04   171.8  1405.4   180.3 1406.73   184.5 1407.62
   188.8 1408.82     210 1415.45   226.9 1421.38   243.9 1427.64   249.1 1429.77
#Mann= 4 ,-1,0
       0     .05       0   68.56    .045       085.83186     .07       0
     130     .06       0
Bank Sta=68.56,85.83186
XS Rating Curve= 0 ,0
Exp/Cntr(USF)=0,0
Exp/Cntr=0.3,0.1

Type RM Length L Ch R = 1 ,7640    ,190.1,202.1,217.1
XS GIS Cut Line= 4
2171109.70913251 712704.865459432171151.25984426 712642.17491187
2171160.73632238712549.5970102422171229.98750864712518.251736463
#Sta/Elev= 30
       0 1405.98    11.7 1405.47    24.6 1405.25      38 1405.41    47.6 1404.38
    66.8 1404.83    71.6 1405.09    76.2 1405.59    80.2 1405.61    84.3 1405.06
    88.3    1403    92.3 1398.11    94.31396.816    96.3 1395.57   100.3 1395.71
     107 1396.82   108.4 1397.02   120.4 1397.36   129.1 1398.35   136.5  1399.3
   152.6 1402.12   164.5 1403.52   171.2 1404.48   176.4  1405.6   180.8 1406.89
   189.6 1409.89   201.4 1414.13   211.6 1417.26   217.8 1419.37   244.3 1429.59
#Mann= 5 ,-1,0
       0     .05       0      60     .07       0    94.3    .045       0
     107     .07       0  165.21     .06       0
Bank Sta=94.3,107
XS Rating Curve= 0 ,0
Exp/Cntr(USF)=0,0
Exp/Cntr=0.3,0.1

Type RM Length L Ch R = 1 ,7438    ,183.9,182,180.2
BEGIN DESCRIPTION:
Structure2 XS1
END DESCRIPTION:
XS GIS Cut Line= 2
2171135.66483252712788.3667393112171344.68014995712730.584822067
#Sta/Elev= 30
       0 1408.69    17.1 1408.07    29.6 1407.34    45.3 1405.47    58.6 1403.53
    71.1 1402.91    75.2    1402    77.8 1400.66    83.5 1397.08    87.5 1396.72
   100.1 1397.39   103.8 1397.15   104.3 1397.09110.15371394.311   112.6 1393.37
   116.7 1393.22   120.9 1393.54123.8536 1394.33   129.2 1395.43   137.5  1396.1
   141.6 1398.06   145.8 1401.79   149.9 1406.03   154.1 1408.37   166.5 1412.97
   170.7 1414.42   175.3 1415.79   183.1 1417.88   198.1 1422.46   216.9 1427.83
#Mann= 4 ,-1,0
       0     .05       0110.1537    .045       0123.8536     .05       0
     170     .06       0
#XS Ineff= 2 , 0
                          354.79         1399.57
Permanent Ineff=
       F       F
Bank Sta=110.1537,123.8536
XS Rating Curve= 0 ,0
Exp/Cntr(USF)=0,0
Exp/Cntr=0.3,0.1

Type RM Length L Ch R = 1 ,7256    ,115.8,116,116.1
BEGIN DESCRIPTION:
Structure3 XS4
END DESCRIPTION:
XS GIS Cut Line= 2
2171206.72915757 712974.136806452171430.37691759712874.763843296
#Sta/Elev= 30
       0  1399.9    10.3 1398.91    19.1 1398.29    41.2 1397.21    71.6  1396.9
      76 1396.17    80.6 1394.22    83.6  1394.1    89.1 1394.33    93.5  1394.3
    97.9 1394.16   101.8 1393.65107.86131391.046     111 1389.97   119.8 1389.69
   128.5 1389.95   132.1 1390.52133.82121391.035   141.6 1394.31     146 1395.25
   154.8 1396.59   165.5 1397.14     181 1397.12   189.8 1397.46   194.2  1398.6
   201.8 1401.74   213.6  1406.3   224.8 1410.19   238.8 1415.71   244.7 1418.59
#Mann= 5 ,-1,0
       0     .05       0     100     .06       0107.8613    .045       0
133.8212     .06       0     210      .1       0
Bank Sta=107.8613,133.8212
XS Rating Curve= 0 ,0
Exp/Cntr(USF)=0,0
Exp/Cntr=0.3,0.1

Type RM Length L Ch R = 1 ,7140    ,42.9,42.8,43.2
BEGIN DESCRIPTION:
Structure3 XS3
END DESCRIPTION:
XS GIS Cut Line= 2
2171246.06088716713075.8894946082171491.75433225712980.147706201
#Sta/Elev= 30
       0 1397.29     6.6 1396.51    10.9 1396.21    40.9 1396.06      71 1394.94
    83.8 1394.62    88.1  1393.9    92.4 1392.52    93.3 1392.39    96.4 1392.26
   109.6 1392.37   113.9 1392.06   122.5 1390.98126.73831390.132   131.1 1389.56
   135.4 1389.48   139.7 1389.72141.42831390.129   152.5 1393.02   156.8 1393.98
   165.4 1395.29   169.7 1395.68     174 1395.89   194.7 1395.51   208.3 1395.05
   212.6 1395.76   216.9 1397.56   242.7 1410.15   250.9 1414.56   263.7 1422.02
#Mann= 4 ,-1,0
       0     .05       0      70     .06       0126.7383    .045       0
141.4283     .06       0
Bank Sta=126.7383,141.4283
XS Rating Curve= 0 ,0
Exp/Cntr(USF)=0,0
Exp/Cntr=0.3,0.1

Type RM Length L Ch R = 1 ,7097    ,216.7,215.8,213.7
BEGIN DESCRIPTION:
Structure3 XS2
END DESCRIPTION:
XS GIS Cut Line= 2
2171262.00323919713114.8596884742171512.02045973713017.784800096
#Sta/Elev= 30
       0 1396.03     6.6 1395.63    28.1 1395.44    49.5 1394.69    79.6 1393.91
    92.4 1394.09    96.7 1392.68     101 1391.76   109.6    1392   123.5 1391.69
   126.8 1391.46133.51151389.986   135.9 1389.46   139.6 1389.12   142.1 1389.11
   148.2 1389.53  149.681389.998   154.4  1391.5   156.8 1392.09   161.1 1392.43
   169.7 1392.62   203.6 1392.16   208.3 1392.32   212.6 1392.97   221.2 1396.64
   229.7 1400.84   234.8 1402.84   238.3 1404.44   259.8 1414.78   268.2 1419.28
#Mann= 5 ,-1,0
       0     .05       0133.5115    .045       0  149.68     .05       0
     180     .06       0     250      .1       0
Bank Sta=133.5115,149.68
XS Rating Curve= 0 ,0
Exp/Cntr(USF)=0,0
Exp/Cntr=0.3,0.1

Type RM Length L Ch R = 1 ,6882    ,295.7,288.5,279.7
BEGIN DESCRIPTION:
Structure3 XS1
END DESCRIPTION:
XS GIS Cut Line= 2
2171376.28150752  713312.52324942171656.75313123 713165.25219615
#Sta/Elev= 30
       0 1398.05     7.2 1394.88    14.2 1392.44    17.2 1391.66    22.5 1390.95
    40.9 1390.57    67.6 1390.44    76.5 1389.95    85.3 1390.56    94.8 1390.43
   108.3 1389.31   117.3 1388.96  122.281388.382   132.7 1387.64   135.4 1387.67
   138.7 1388.39   144.5 1389.81   153.5 1390.19   171.3 1389.34   206.8 1388.86
   221.6 1388.37   248.3 1389.03   261.9 1388.85   266.4 1389.04     271 1390.25
   274.9 1392.02   282.5 1394.49   295.7 1400.49   307.1  1406.5   316.8 1412.26
#Mann= 4 ,-1,0
       0      .1       0  122.28    .045       0   138.7      .1       0
     140     .06       0
#XS Ineff= 2 , 0
           85.86 1392.66
Permanent Ineff=
       F       F
Bank Sta=122.28,138.7
XS Rating Curve= 0 ,0
Exp/Cntr(USF)=0,0
Exp/Cntr=0.3,0.1

Type RM Length L Ch R = 1 ,6593    ,258.7,265.4,266.5
XS GIS Cut Line= 3
2171554.98885414713529.0023011642171662.08295634713369.711073515
2171729.57923925713229.318805079
#Sta/Elev= 30
       0 1436.77     4.6 1435.73    16.5 1431.75      38 1422.13    43.2 1419.22
    46.8 1416.64    61.3 1404.56    72.1 1394.87    73.8 1393.59    76.9 1391.95
     101 1391.49   124.7 1392.54   136.2 1392.49   178.1 1391.07   188.5 1390.23
   219.2 1388.85   241.4 1387.35  246.041386.749   250.2 1385.86   254.7 1385.57
   263.5 1385.83  267.351386.766   272.4 1388.56   280.8 1390.38   307.6 1391.88
   319.8 1393.57   325.7 1396.04   330.1 1398.57     339 1402.75   347.7 1406.05
#Mann= 5 ,-1,0
       0      .1       0      70     .06       0  246.04    .045       0
  267.35     .06       0  331.94      .1       0
Bank Sta=246.04,267.35
XS Rating Curve= 0 ,0
Exp/Cntr(USF)=0,0
Exp/Cntr=0.3,0.1

Type RM Length L Ch R = 1 ,6328    ,299.2,309.1,315.9
XS GIS Cut Line= 3
2171718.69258196713630.1553711982171935.30400671713406.496669927
 2171927.5752115713300.878050797
#Sta/Elev= 30
       0 1407.02     4.6 1404.58    23.6  1396.1    30.9 1391.76    34.8 1390.58
      47 1390.97    65.4 1390.12    90.5 1390.68   112.7 1389.49   157.3 1388.22
   191.9 1388.82   225.2 1388.82   240.8 1388.36   257.5 1386.41   263.1 1385.02
   266.6 1384.11   272.4 1383.75   278.1  1384.2   280.41385.072   289.6 1391.79
   295.4 1394.51   301.1 1395.26   332.7 1397.65   341.7 1398.88   360.8 1403.39
   376.9 1406.15   386.5 1408.67   400.9 1410.52   408.9 1412.68   417.3  1415.6
#Mann= 7 ,-1,0
       0     .05       0     110     .06       0     130     .07       0
     250     .08       0     260      .1       0   263.1    .045       0
   280.4      .1       0
#XS Ineff= 2 , 0
          141.36 1394.26
Permanent Ineff=
       F       F
Bank Sta=263.1,280.4
XS Rating Curve= 0 ,0
Exp/Cntr(USF)=0,0
Exp/Cntr=0.3,0.1

Type RM Length L Ch R = 1 ,6019    ,171.7,172.4,172.5
XS GIS Cut Line= 2
2171825.16229158713726.1285331712172125.70780407 713686.44977169
#Sta/Elev= 30
       0 1407.14     7.1 1404.13    21.4 1398.77    24.9 1397.02      32 1392.75
    35.6 1391.15    39.2 1390.86    47.4 1391.42    59.5 1391.28    67.7 1390.96
    75.7 1390.07    89.1 1389.82   135.4 1390.19   160.4 1389.97   172.5 1389.11
   188.6 1386.21   216.9  1384.2   220.9 1382.89   220.9 1382.87   224.9 1381.91
     229 1381.81     233 1382.39  234.081382.906   237.1 1384.32   238.8 1385.68
     253 1398.82   257.2    1402   263.7 1405.27   288.7 1415.35   303.2 1422.73
#Mann= 5 ,-1,0
       0     .05       0      70     .06       0     170     .07       0
   220.9    .045       0  234.08     .07       0
Bank Sta=220.9,234.08
XS Rating Curve= 0 ,0
Exp/Cntr(USF)=0,0
Exp/Cntr=0.3,0.1

Type RM Length L Ch R = 1 ,5846    ,229.2,248.3,268
BEGIN DESCRIPTION:
Structure4 XS4
END DESCRIPTION:
XS GIS Cut Line= 2
2171877.57989044 713884.491270162172135.06972558713860.852859066
#Sta/Elev= 30
       0 1415.83    14.7 1409.13    22.7  1404.3    30.7 1398.24    34.7 1397.12
    54.8  1396.4    58.8 1395.88    66.9 1394.24    74.9 1393.46    78.9 1393.44
     103 1394.53   115.1 1394.35   127.1 1393.25   159.3 1389.43   163.3 1389.18
   167.3 1388.05   175.3 1381.66  176.191381.289   179.3 1379.93   183.4 1379.83
   187.4 1380.11  192.371381.273   195.4    1382   203.4 1385.74   215.5 1390.45
   219.5 1392.69   231.6 1400.69   239.6 1405.49   255.7 1417.48   258.6 1419.12
#Mann= 4 ,-1,0
       0     .06       0  176.19    .045       0  192.37     .06       0
     210     .07       0
Bank Sta=176.19,192.37
XS Rating Curve= 0 ,0
Exp/Cntr(USF)=0,0
Exp/Cntr=0.3,0.1

Type RM Length L Ch R = 1 ,5598    ,46.2,44.6,47.2
BEGIN DESCRIPTION:
Structure4 XS3
END DESCRIPTION:
XS GIS Cut Line= 5
2171878.42411941713916.5719709322171984.79696933 713906.44122332
2171990.70657211714022.1005918912172029.54110462714195.167530265
2172108.89862758 714174.90603504
#Sta/Elev= 30
       0 1410.84    21.8 1400.23    25.9 1398.67    33.9 1397.45      50 1396.87
    74.1  1393.8   106.9 1394.25   133.6 1393.47   197.7 1387.37   222.7  1386.7
   247.6 1384.95   266.6 1384.87   283.2 1379.57  293.831377.222   303.5 1375.99
  312.331377.245   320.7 1380.93   336.5 1390.65   348.8 1396.24   352.9 1397.12
   381.6 1396.29     400 1396.92   406.9  1404.1     411 1409.84   413.7 1412.54
   419.3 1415.87   435.8 1421.15   460.5 1426.61   472.9  1430.9   481.9  1432.2
#Mann= 4 ,-1,0
       0     .06       0  293.83    .045       0  312.33     .06       0
  460.03      .1       0
Bank Sta=293.83,312.33
XS Rating Curve= 0 ,0
Exp/Cntr(USF)=0,0
Exp/Cntr=0.3,0.1

Type RM Length L Ch R = 1 ,5553    ,240.4,219.7,182.4
BEGIN DESCRIPTION:
Structure4 XS2
END DESCRIPTION:
XS GIS Cut Line= 5
2171843.38861725713945.2757558332171949.76146717713935.145008221
2171955.67106995714050.8043767922171994.50560246714223.871315166
2172073.86312542714203.609819941
#Sta/Elev= 30
       0 1411.57    36.3 1404.72      49    1403   101.2 1393.66   136.9 1392.15
   179.7 1392.02     201 1389.72     221 1389.12   245.6 1385.53   265.3 1383.61
     282 1380.93   293.8 1376.28   298.9 1375.12   311.2 1375.38  316.651376.285
   322.2 1378.51   332.2  1385.7     344 1389.87   368.6 1391.89     400 1390.36
   405.9 1393.59     410  1394.9   422.4 1395.39   438.9 1395.07   443.1 1397.48
   451.3 1408.34   456.2 1413.27   459.4  1415.3   463.7 1417.08   481.9 1422.38
#Mann= 6 ,-1,0
       0     .05       0      90     .06       0  116.85     .05       0
   293.8    .045       0  316.65     .05       0  362.66     .06       0
Bank Sta=293.8,316.65
XS Rating Curve= 0 ,0
Exp/Cntr(USF)=0,0
Exp/Cntr=0.3,0.1

Type RM Length L Ch R = 1 ,5334    ,142.3,147.6,150
BEGIN DESCRIPTION:
Structure4 XS1
END DESCRIPTION:
XS GIS Cut Line= 2
2171896.85692539714352.9880949442172075.33537144714242.208369806
#Sta/Elev= 30
       0 1408.52    16.8 1399.02    27.4 1396.18    41.6 1388.68    51.7 1381.18
    60.4 1370.73    63.3 1369.25    66.2 1368.37    69.8 1367.96    79.2 1368.37
    88.6  1368.6    93.4 1369.94    98.1  1372.3   102.8 1374.05   112.2 1379.32
   116.9 1381.05   128.6 1383.88   136.2  1387.1   141.7 1389.95   150.4  1396.2
   154.6 1397.99   159.3 1398.69   166.5 1399.01   176.6 1398.85   182.8 1398.25
   187.5 1400.78   192.2 1405.47   196.9 1409.27   204.4 1413.55   210.1 1415.76
#Mann= 3 ,-1,0
       0     .05       0    66.2    .045       0    79.2     .05       0
Bank Sta=66.2,79.2
XS Rating Curve= 0 ,0
Exp/Cntr(USF)=0,0
Exp/Cntr=0.3,0.1

Type RM Length L Ch R = 1 ,5186    ,149.2,154.7,158.1
XS GIS Cut Line= 2
2171960.21451441714456.2467011732172099.35458164714419.658886424
#Sta/Elev= 30
       0 1388.69     4.1 1386.27     8.2 1384.22       9 1383.97    12.4 1383.12
    20.6 1381.99    37.2 1377.32    41.3 1376.04    45.5 1374.53    49.6 1372.34
    61.4 1365.08   65.951363.453    70.3 1362.35    74.4 1362.06    78.5 1363.05
    81.1 1363.47    82.7 1363.65    86.8 1365.32      91 1369.63    96.6 1377.34
    99.2 1380.76   103.4 1384.32   107.5 1385.99   111.6 1385.95   115.8 1386.31
   119.9 1388.23     124 1391.36   128.2 1394.92   140.6 1406.21   143.9  1408.8
#Mann= 6 ,-1,0
       0     .05       0      30      .1       0   65.95    .045       0
    81.1      .1       0     110     .05       0     130      .1       0
Bank Sta=65.95,81.1
XS Rating Curve= 0 ,0
Exp/Cntr(USF)=0,0
Exp/Cntr=0.3,0.1

Type RM Length L Ch R = 1 ,5031    ,144.8,146.1,146.5
XS GIS Cut Line= 3
2171989.84695118 714586.933345372172128.89146215714582.374508944
 2172156.2444807714617.325588206
#Sta/Elev= 30
       0 1380.82     2.3 1379.68     6.3 1378.22    10.3 1377.25    22.3 1375.34
    27.2 1374.05    30.3 1372.78    34.3 1370.36    42.4 1363.45    46.4 1360.33
    50.4 1358.47    58.4 1356.31   63.521355.331    70.4 1354.54    82.4 1354.08
    86.4 1354.28    90.4 1354.96   91.091355.339    94.4 1357.17    98.4 1360.41
   106.4 1364.29   118.4 1371.26   122.4 1375.37   126.4    1378   130.4 1379.03
   142.7 1380.32   154.9 1382.37   160.6 1383.66   169.1 1386.24   183.5 1389.08
#Mann= 3 ,-1,0
       0      .1       0   63.52    .045       0   91.09      .1       0
Bank Sta=63.52,91.09
XS Rating Curve= 0 ,0
Exp/Cntr(USF)=0,0
Exp/Cntr=0.3,0.1

Type RM Length L Ch R = 1 ,4885    ,165,173.9,182.9
XS GIS Cut Line= 2
2171964.46212363714728.2788416542172127.06062281714730.558259867
#Sta/Elev= 30
       0 1375.81     7.7 1373.96    15.7 1372.73    19.7 1371.48    23.7 1369.63
    31.7 1365.03    35.7 1362.93    39.7 1361.12    43.7 1359.76    47.7 1359.11
    59.7 1358.35    67.7 1357.28    71.7 1356.99    75.7 1356.06    83.7 1352.69
   85.041352.371    87.7 1351.71    91.7 1351.56   103.7 1351.69   115.7 1352.42
   119.7 1354.28   124.6 1358.62   127.7 1361.54   130.8 1364.85   139.7 1375.02
   143.7  1378.7   147.7 1382.63   151.7 1386.33   154.5 1388.73   162.6 1396.33
#Mann= 3 ,-1,0
       0      .1       0   85.04    .045       0   115.7      .1       0
Bank Sta=85.04,115.7
XS Rating Curve= 0 ,0
Exp/Cntr(USF)=0,0
Exp/Cntr=0.3,0.1

Type RM Length L Ch R = 1 ,4711    ,147.9,141.7,134.2
XS GIS Cut Line= 2
2171950.76517557714862.0601759772172066.91771738714921.382718789
#Sta/Elev= 30
       0 1371.26     6.1 1370.87    10.6 1370.41    15.1 1369.68    19.5 1367.93
    30.1 1361.37      33 1359.49    37.5 1356.29    46.5 1348.11      51 1345.99
    53.9 1345.45      60 1344.59    64.5 1344.32    68.8  1344.4    73.4 1344.88
    77.7 1345.12    80.51345.457    82.4 1345.77    86.9  1347.3    89.6 1348.89
    91.4 1350.09    95.9 1354.09   100.4    1357   104.9 1359.59   110.4 1364.33
   112.4 1365.94   118.4 1370.06   125.3 1375.15   127.3 1376.81   130.4 1378.94
#Mann= 3 ,-1,0
       0      .1       0    53.9    .045       0    80.5      .1       0
Bank Sta=53.9,80.5
XS Rating Curve= 0 ,0
Exp/Cntr(USF)=0,0
Exp/Cntr=0.3,0.1

Type RM Length L Ch R = 1 ,4570    ,166.9,170.9,173
XS GIS Cut Line= 2
2171880.34311552715018.4690500712172070.29463325715035.353629425
#Sta/Elev= 30
       0 1364.94     3.8 1362.74    15.9 1354.79    19.9 1352.66    23.9 1351.43
      44 1348.75      48 1348.82      52 1349.65    56.1 1350.07    60.1 1348.57
    64.1  1344.8    68.1 1342.26    72.1 1341.31   75.131340.972    84.2 1340.36
    96.2 1340.47   100.2 1341.02   104.2    1342   108.3 1342.63   112.3 1342.91
   124.3 1342.53   132.4 1343.99   144.4 1345.57   148.4 1347.31   156.4 1351.94
   164.6 1358.25   168.7 1361.11   175.7 1365.03   184.6 1370.38   190.7 1374.75
#Mann= 3 ,-1,0
       0      .1       0   75.13    .045       0   100.2      .1       0
Bank Sta=75.13,100.2
XS Rating Curve= 0 ,0
Exp/Cntr(USF)=0,0
Exp/Cntr=0.3,0.1

Type RM Length L Ch R = 1 ,4399    ,256.8,253.9,250.2
XS GIS Cut Line= 2
2171884.56426036715172.1187221892172008.66591861715210.953254702
#Sta/Elev= 30
       0 1366.77     3.8 1365.93       8 1363.95    19.7 1359.43    22.9 1357.81
    24.7 1356.72    33.1 1347.99    37.3 1344.34    41.5 1341.57    45.7 1339.47
    54.1 1338.02    58.3 1336.73   63.031336.207      74 1335.48    79.2 1335.36
   82.141336.251    83.4 1336.68    86.7 1338.88    89.9 1341.53    91.8 1343.22
    93.1 1344.52      96 1347.54    99.5 1352.09   104.4 1358.77   105.9 1360.62
   112.3    1368   116.9 1373.04   121.8 1377.97   125.3    1381     130 1384.79
#Mann= 3 ,-1,0
       0      .1       0   63.03    .045       0   82.14      .1       0
Bank Sta=63.03,82.14
XS Rating Curve= 0 ,0
Exp/Cntr(USF)=0,0
Exp/Cntr=0.3,0.1

Type RM Length L Ch R = 1 ,4145    ,195.6,186.6,173.4
XS GIS Cut Line= 3
2171794.20954314715417.4168553552171926.58701573 715436.84730353
2171985.68304347715398.856999985
#Sta/Elev= 30
       0 1383.52       2 1381.99       6 1378.33    10.1 1374.01    14.1 1370.21
    22.7  1363.2    26.2 1360.01    42.4 1343.76    50.5 1337.71    54.5  1334.3
    57.9 1332.19    58.6 1331.84    62.6 1331.43    82.8 1330.47    86.9  1330.6
   92.321331.468      95 1332.22      99 1333.87   106.9  1337.9   115.2 1342.59
   119.2 1344.19   123.3 1344.97   133.8 1345.38   154.7 1343.33   160.8 1343.62
   166.8 1345.12   178.1  1349.4   183.2 1350.91   197.5 1354.04     204 1354.75
#Mann= 3 ,-1,0
       0      .1       0    62.6    .045       0   92.32      .1       0
Bank Sta=62.6,92.32
XS Rating Curve= 0 ,0
Exp/Cntr(USF)=0,0
Exp/Cntr=0.3,0.1

Type RM Length L Ch R = 1 ,3958    ,194.9,195.5,195.1
XS GIS Cut Line= 2
2171863.70759151715625.7148729532172102.38467002715507.939720672
#Sta/Elev= 30
       0 1356.26     6.7 1350.56    13.9 1344.07    27.3 1334.48    30.6 1331.16
   35.59 1327.01    36.2  1326.5    40.7 1325.31    45.1 1325.12    49.6 1325.42
      54 1326.04    57.5 1327.01      63 1328.83    67.4 1329.46    81.4 1330.77
    94.2 1332.27   107.6 1332.25   116.5 1334.36     121 1334.96   127.8 1335.23
   152.2 1337.44     170 1340.47   187.9 1342.19   196.8 1343.94   210.2 1347.88
   214.6 1348.65   223.5 1349.61   241.4 1352.13   254.8 1354.56   266.2 1357.31
#Mann= 4 ,-1,0
       0     .05       0      30      .1       0   35.59    .045       0
    57.5      .1       0
Bank Sta=35.59,57.5
XS Rating Curve= 0 ,0
Exp/Cntr(USF)=0,0
Exp/Cntr=0.3,0.1

Type RM Length L Ch R = 1 ,3763    ,202.1,212,207.1
XS GIS Cut Line= 2
 2171953.3417782715798.7296984282172149.28627934715700.757447858
#Sta/Elev= 30
       0 1340.75     6.2 1336.45     9.2 1334.75    21.2 1330.11      30 1325.52
    34.5 1323.79    38.9 1323.16    43.4 1323.11    61.3  1323.4    65.8 1323.78
    74.7 1325.11    88.1  1324.8    97.1 1324.08   101.7 1324.25     106 1325.09
   107.6 1325.83   110.5 1327.51     115 1330.96   116.6 1331.87   119.4 1333.19
   122.5 1334.06   125.5 1334.47   137.3 1334.59   155.5  1335.8   164.2 1336.56
   177.6 1338.76   188.1 1341.23   204.4 1346.39     209 1348.47   219.1 1354.59
#Mann= 3 ,-1,0
       0      .1       0    34.5    .045       0    65.8      .1       0
Bank Sta=34.5,65.8
XS Rating Curve= 0 ,0
Exp/Cntr(USF)=0,0
Exp/Cntr=0.3,0.1

Type RM Length L Ch R = 1 ,3551    ,162.9,166.9,168.5
XS GIS Cut Line= 2
2171993.72250043715974.7571706072172216.64960164715892.698114949
#Sta/Elev= 30
       0 1342.99    11.1 1335.29    19.7 1330.89    23.9 1329.39    28.2 1328.48
    45.2  1326.2    53.8 1323.61      58 1322.72    62.3 1322.34    74.8 1322.34
    87.3 1321.49    93.5 1321.43    96.6 1320.98   100.6 1319.55  106.911318.503
   113.4 1317.72   117.7 1317.67   126.2 1318.05  128.921318.492   130.5 1318.76
     134 1320.95   140.2 1326.74   143.3 1328.99   146.5 1330.53   151.8  1331.7
   173.1 1334.66   177.4  1335.7   198.7 1345.46   227.5 1363.08   237.6 1369.71
#Mann= 3 ,-1,0
       0      .1       0  106.91    .045       0  128.92      .1       0
Bank Sta=106.91,128.92
XS Rating Curve= 0 ,0
Exp/Cntr(USF)=0,0
Exp/Cntr=0.3,0.1

Type RM Length L Ch R = 1 ,3384    ,190.5,187,184.6
XS GIS Cut Line= 2
2172024.96458628716118.3733352092172231.68849471716074.875675852
#Sta/Elev= 30
       0 1339.86    11.5 1334.03    19.6 1330.78    25.2 1329.14      36 1326.66
    48.2 1325.11    56.4 1323.42    60.5 1322.01    68.7 1318.57    72.8 1318.34
    80.9  1319.6    97.3 1320.41   101.4 1319.73   106.1 1317.69   109.6 1317.02
   125.9 1316.46   138.2 1316.63   142.3 1317.69   146.3 1319.26   154.5 1318.97
   158.6 1319.41   162.7 1321.71   166.8 1325.54   170.9  1328.9     175 1331.38
     179 1334.28   187.2 1341.08   194.2 1348.02   203.6 1358.42   211.3 1367.42
#Mann= 3 ,-1,0
       0      .1       0   106.1    .045       0   142.3      .1       0
#XS Ineff= 2 , 0
           87.46 1325.32
Permanent Ineff=
       F       F
Bank Sta=106.1,142.3
XS Rating Curve= 0 ,0
Exp/Cntr(USF)=0,0
Exp/Cntr=0.3,0.1

Type RM Length L Ch R = 1 ,3197    ,318.5,334.8,356
XS GIS Cut Line= 2
2172056.75862441716324.9414458742172298.14901314716235.360310114
#Sta/Elev= 30
       0 1346.03     7.9 1341.45    20.7 1335.58      25 1333.73    30.5 1332.08
      46 1329.43    63.4 1325.77    76.2 1322.35    80.4 1321.99    97.5 1321.53
   123.1 1321.88   126.9 1321.61   127.4 1321.51   131.6 1318.89   135.9 1315.44
   139.4 1313.85  141.31 1313.45   157.2 1312.58   165.8 1313.46   174.3 1314.85
   187.1 1314.85   191.4 1315.44   195.4 1316.37   199.9 1317.95   206.3  1320.9
   212.7 1324.36   221.2 1329.52     234    1336   250.4 1345.49   257.5  1348.5
#Mann= 3 ,-1,0
       0      .1       0  141.31    .045       0   165.8      .1       0
Bank Sta=141.31,165.8
XS Rating Curve= 0 ,0
Exp/Cntr(USF)=0,0
Exp/Cntr=0.3,0.1

Type RM Length L Ch R = 1 ,2862    ,186.6,182.7,177.2
XS GIS Cut Line= 2
2172062.32436311716462.230805985 2172227.2022805716593.677256252
#Sta/Elev= 30
       0 1338.43     2.4 1337.67    11.1  1335.6    26.2 1331.52    43.3 1326.65
    48.4 1325.58    51.8 1324.67    63.8 1320.68    68.9 1319.28      74 1318.82
    79.1  1318.6    89.3 1316.95     101 1315.63   107.4 1313.75   111.6 1311.63
   114.4 1310.48   120.1 1309.57   125.1 1309.55   128.7 1309.21   134.3 1308.03
   140.5 1307.51   150.7 1307.85     160  1307.6  165.261308.031   171.4 1309.08
     178 1313.08   181.4 1314.87   186.5 1316.61   194.1 1319.71   210.9 1324.97
#Mann= 3 ,-1,0
       0      .1       0   134.3    .045       0  165.26      .1       0
Bank Sta=134.3,165.26
XS Rating Curve= 0 ,0
Exp/Cntr(USF)=0,0
Exp/Cntr=0.3,0.1

Type RM Length L Ch R = 1 ,2679    ,164.5,159.5,151.2
XS GIS Cut Line= 2
2172018.75068354716675.8998306082172186.67002554716748.857889543
#Sta/Elev= 30
       0 1339.16    17.3 1329.07    26.4 1323.35    29.4 1321.05    32.5  1318.2
    35.5 1313.38    38.5 1308.27    40.8 1304.88   41.511304.516    45.2 1303.45
    50.7 1303.38    62.6 1303.92      67 1304.61    80.1  1307.4    84.1 1308.01
   102.4  1308.4   110.6 1309.03   119.3 1309.39   123.7 1310.66     128  1313.6
   132.4 1316.19   135.8 1317.35   143.7 1319.54   149.8 1320.57   160.1 1323.88
   162.9 1324.47   171.6 1325.11   175.4 1325.88   178.4 1327.36   183.1 1330.25
#Mann= 3 ,-1,0
       0      .1       0   41.51    .045       0      67      .1       0
Bank Sta=41.51,67
XS Rating Curve= 0 ,0
Exp/Cntr(USF)=0,0
Exp/Cntr=0.3,0.1

Type RM Length L Ch R = 1 ,2520    ,261.1,267.3,253.5
XS GIS Cut Line= 2
2171964.07127926716849.055596113 2172175.9970695716846.739467258
#Sta/Elev= 30
       0 1340.11     8.1 1332.47    12.1 1329.21    16.1 1326.36    24.1  1321.6
    28.1 1318.81    36.1    1312    40.1 1307.94    44.1 1304.99    48.1 1303.91
    56.9 1302.83    68.1 1302.06    72.1 1302.17    76.1 1302.81    80.1 1304.02
    84.1 1304.72    88.1 1304.85    96.1 1304.71   120.1 1303.18   124.1 1303.39
   128.1 1304.28   132.1 1305.94   140.1 1310.84   144.1 1312.72   152.1 1314.06
   156.1 1315.36   184.1 1326.01   200.1 1333.99   208.1 1339.23   211.9 1341.05
#Mann= 3 ,-1,0
       0      .1       0    56.9    .045       0    76.1      .1       0
Bank Sta=56.9,76.1
XS Rating Curve= 0 ,0
Exp/Cntr(USF)=0,0
Exp/Cntr=0.3,0.1

Type RM Length L Ch R = 1 ,2253    ,201,205.7,211.4
XS GIS Cut Line= 3
2172042.92670856 717058.277919922172081.85123588717032.504200498
2172244.69743184 717023.90539077
#Sta/Elev= 30
       0 1322.95     6.3 1318.91    11.1 1316.41    20.7 1312.41      31 1308.99
    35.1 1307.28    44.7 1300.95    46.7 1300.29    55.9 1299.21      61 1299.33
      69 1300.28    85.1  1299.6    97.1 1298.49   109.1 1298.78   113.1 1298.05
   117.1 1296.73   121.1 1296.04   125.1 1296.03     132 1296.74   141.1 1297.79
   153.2 1297.82   157.2 1298.15   161.2 1300.65   165.2 1304.83   169.2    1308
   181.4 1314.99   189.2  1320.2   193.2 1323.74   205.2 1335.73   209.8 1339.72
#Mann= 3 ,-1,0
       0      .1       0   117.1    .045       0     132      .1       0
Bank Sta=117.1,132
XS Rating Curve= 0 ,0
Exp/Cntr(USF)=0,0
Exp/Cntr=0.3,0.1

Type RM Length L Ch R = 1 ,2047    ,143.1,142.4,141.5
XS GIS Cut Line= 2
2172080.66433438717198.1218313072172250.52657959717249.819036371
#Sta/Elev= 30
       0 1323.97    16.2 1315.69    20.4 1312.51    24.6 1308.18    28.8 1304.18
    32.9 1300.91    41.3 1295.61    45.5 1294.14    46.9 1293.99    49.7 1293.82
    70.6 1293.85    74.7 1293.55   82.461291.126    87.3 1290.38    91.5 1290.34
    99.8 1290.61   101.4 1291.15     104 1292.08   108.2 1294.38   127.1 1306.84
   130.3 1308.68   133.3 1309.95   137.5 1310.95   141.6 1312.31   145.8 1314.39
     150 1316.15   158.4 1318.56   162.6 1320.15   170.9 1324.14   177.6    1328
#Mann= 3 ,-1,0
       0      .1       0   82.46    .045       0   101.4      .1       0
Bank Sta=82.46,101.4
XS Rating Curve= 0 ,0
Exp/Cntr(USF)=0,0
Exp/Cntr=0.3,0.1

Type RM Length L Ch R = 1 ,1905    ,190,182.3,173.6
XS GIS Cut Line= 2
2172053.28570755717343.7799382132172223.06953327717383.177290038
#Sta/Elev= 30
       0  1341.3     3.6 1337.22    10.2 1330.99    23.5 1321.24    31.7 1312.88
    35.8 1308.26    36.9 1306.64    39.9 1301.78    41.6 1298.45      44 1293.38
    48.1 1289.26    52.2 1288.56    60.5 1288.83    64.6 1289.25    68.7 1289.17
    71.5 1288.86    76.9 1288.44   82.581288.847    93.3 1290.72   101.5 1291.19
   105.6 1291.73   113.8 1293.38     122 1294.72   126.2 1296.36   134.4 1301.87
   136.9 1303.21   142.6 1305.54   150.8 1307.32   163.1 1310.37   174.3 1314.35
#Mann= 3 ,-1,0
       0      .1       0    71.5    .045       0   82.58      .1       0
Bank Sta=71.5,82.58
XS Rating Curve= 0 ,0
Exp/Cntr(USF)=0,0
Exp/Cntr=0.3,0.1

Type RM Length L Ch R = 1 ,1722    ,202.9,203.5,200.7
XS GIS Cut Line= 2
2172035.57481564717555.299442394 2172228.2084488717506.679451916
#Sta/Elev= 30
       0 1310.52     5.5 1308.42      13  1306.3    28.6 1303.71    33.6 1302.59
    41.4 1300.09    50.1 1296.58    54.2 1295.55    62.5 1294.02    66.6 1292.58
      79 1286.36   82.051285.413    83.1 1285.11    87.3 1284.67    99.6 1284.41
   107.9  1284.6   124.4 1285.41   128.5 1286.45   132.6  1289.9   137.3 1294.86
   140.6 1297.67   143.9 1300.12   149.1 1303.32   157.4 1307.61   165.6 1312.38
   170.2  1314.8   182.1 1319.89   186.3 1321.96   190.4 1324.19   198.7 1329.27
#Mann= 3 ,-1,0
       0      .1       0   82.05    .045       0   124.4      .1       0
Bank Sta=82.05,124.4
XS Rating Curve= 0 ,0
Exp/Cntr(USF)=0,0
Exp/Cntr=0.3,0.1

Type RM Length L Ch R = 1 ,1519    ,175.2,179.3,183.6
XS GIS Cut Line= 2
2172086.10510867717745.0360569482172265.81444056717686.568979791
#Sta/Elev= 30
       0 1305.52     6.4 1303.44    14.8 1301.21      19 1300.45      40 1298.11
    48.4 1296.33    52.7 1295.14    65.3 1288.66    69.5 1285.76    73.7 1283.19
   79.42 1281.16    82.1 1280.32    86.3 1279.65    90.5 1279.62    98.9 1280.05
   107.3 1281.15   111.5 1283.28   115.7 1286.62     120 1290.59   124.2 1294.11
   128.4 1296.87   132.6  1299.2   145.2 1305.66   149.4 1308.27     162 1317.28
   165.6 1320.28   169.7 1324.33   182.4 1337.99   185.6 1340.66     189 1342.94
#Mann= 3 ,-1,0
       0      .1       0   79.42    .045       0   107.3      .1       0
Bank Sta=79.42,107.3
XS Rating Curve= 0 ,0
Exp/Cntr(USF)=0,0
Exp/Cntr=0.3,0.1

Type RM Length L Ch R = 1 ,1339    ,220.5,227,233.9
XS GIS Cut Line= 2
2172112.29421688717899.916990113 2172301.0300449717882.137528054
#Sta/Elev= 30
       0 1311.58     3.9 1309.18     7.9 1307.14      16 1303.51      24 1299.36
      32  1296.6    40.1 1292.34    45.6 1290.45    52.1 1288.63    60.1  1287.6
    64.2 1286.59    68.2 1284.88    76.2 1279.52   86.571276.837    92.3 1275.91
    96.3 1275.81   104.3 1276.03   116.4 1276.97   120.4 1278.07   128.4 1284.16
   136.5 1287.53   148.5 1293.26   156.5 1297.72   160.9 1299.81   172.6 1304.66
   176.7 1306.64   180.7 1309.44   184.7 1312.89   188.7 1317.04   189.6  1318.2
#Mann= 3 ,-1,0
       0      .1       0   86.57    .045       0   116.4      .1       0
Bank Sta=86.57,116.4
XS Rating Curve= 0 ,0
Exp/Cntr(USF)=0,0
Exp/Cntr=0.3,0.1

Type RM Length L Ch R = 1 ,1112    ,151.6,154.9,158.5
XS GIS Cut Line= 2
2172125.45033833718088.1342716192172298.68612249718136.761860157
#Sta/Elev= 30
       0 1302.08     3.1 1301.26      16 1297.11    18.7 1295.95    23.6  1292.9
    27.8 1290.53    32.3 1287.72    36.1 1284.81    40.2 1280.76    44.4 1276.28
    48.5 1272.96    48.5 1272.92    52.7 1271.43    56.8 1271.07      61 1271.23
    65.1 1271.79    73.5 1271.88    77.6  1272.5   78.881272.965    81.8 1274.13
    85.9 1276.49    90.6 1277.82   135.8 1279.42   144.1 1279.39     149 1279.81
   152.4 1280.67   156.6 1282.64   166.7 1288.02   173.2 1291.98   179.9 1296.49
#Mann= 3 ,-1,0
       0      .1       0    48.5    .045       0   78.88      .1       0
Bank Sta=48.5,78.88
XS Rating Curve= 0 ,0
Exp/Cntr(USF)=0,0
Exp/Cntr=0.3,0.1

Type RM Length L Ch R = 1 ,958     ,131,133.9,139.1
XS GIS Cut Line= 2
2172086.12535266718223.7540129292172274.38841245718323.373031115
#Sta/Elev= 30
       0 1298.17     2.3 1296.39     5.5 1294.41    15.9 1289.22    17.4 1288.21
    26.2 1281.22    29.2 1279.21      34 1276.55    37.3 1274.09      43 1269.21
    47.6 1268.24    55.8 1268.41    56.6 1268.49    58.8 1269.22    61.2 1270.13
    65.7 1272.91    70.2 1274.18    71.5 1274.27    88.4  1274.5   112.1 1274.32
   151.7 1274.87   165.3 1274.82   169.8  1276.1   177.2 1280.15   182.6 1283.33
   196.9 1290.13   200.9 1291.77   203.8 1293.24     206  1294.4     213 1299.06
#Mann= 3 ,-1,0
       0      .1       0      43    .045       0    58.8      .1       0
Bank Sta=43,58.8
XS Rating Curve= 0 ,0
Exp/Cntr(USF)=0,0
Exp/Cntr=0.3,0.1

Type RM Length L Ch R = 1 ,824     ,175.9,179.9,180.2
XS GIS Cut Line= 2
2172022.80818009718329.2826338892172194.18666052718467.736184589
#Sta/Elev= 30
       0 1306.17     1.8 1305.09     6.9 1301.42     9.4 1299.18    17.2 1291.61
    22.3 1286.23    42.9 1268.43    44.81267.246    46.4 1266.55      48 1266.14
    57.8 1265.88    69.2 1266.12      72 1266.48    74.9 1267.31    78.9 1268.95
    80.5 1269.36    83.4 1269.71   125.2 1269.65   152.6 1270.97     156 1271.28
   161.2 1272.11   165.9 1273.36   171.5 1275.22   186.9 1281.06   190.8 1282.82
     200  1287.5   207.4 1290.73   211.4 1292.77   212.6 1293.48   220.3 1299.12
#Mann= 3 ,-1,0
       0      .1       0    44.8    .045       0    74.9      .1       0
#XS Ineff= 2 , 0
                           83.88          1272.5
Permanent Ineff=
       F       F
Bank Sta=44.8,74.9
XS Rating Curve= 0 ,0
Exp/Cntr(USF)=0,0
Exp/Cntr=0.3,0.1

Type RM Length L Ch R = 1 ,644     ,171.2,174,174.9
XS GIS Cut Line= 2
  2171910.192907718450.777389066 2172053.7962544718608.057245745
#Sta/Elev= 30
       0 1289.21     8.8  1284.9    11.6 1282.89    14.8 1280.22    19.5 1276.61
    22.9 1274.22    25.8 1271.89    31.4 1267.02    34.2 1264.85    35.8 1263.85
    38.5 1262.67    41.2 1262.09    46.6 1261.81    62.6 1262.31    65.4 1262.65
    73.7    1264    80.1 1264.31    85.2  1265.3    91.9 1265.98   115.7 1266.67
   130.5 1266.79   163.1 1268.58   170.2 1269.47   176.6 1269.07     182 1269.47
   187.4 1270.97   192.8 1274.51   198.2 1279.63   204.6  1284.8     213 1291.12
#Mann= 3 ,-1,0
       0      .1       0    38.5    .045       0    65.4      .1       0
Bank Sta=38.5,65.4
XS Rating Curve= 0 ,0
Exp/Cntr(USF)=0,0
Exp/Cntr=0.3,0.1

Type RM Length L Ch R = 1 ,470     ,150.4,169.9,179.1
XS GIS Cut Line= 2
2171773.54466294 718539.731444522171919.46078081718738.918526058
#Sta/Elev= 30
       0 1297.69    11.2 1290.54    34.4 1274.85    41.5 1270.24    46.4 1266.59
    54.4 1259.64    56.3 1258.59    57.3 1258.39   66.24 1257.47    71.2 1256.87
    74.5 1256.79    81.1 1256.86    85.7 1257.49    92.4 1260.29      96 1260.86
     101 1260.92   120.8 1260.46   125.8  1260.7   130.7 1261.22   175.3  1264.3
   186.1 1265.38   194.7 1265.91   207.5 1267.24   211.8 1268.93   214.3 1270.34
   220.4  1274.6   224.9    1277   227.8 1278.11   240.5 1281.11   246.9 1283.32
#Mann= 5 ,-1,0
       0      .1       0   66.24    .045       0    85.7      .1       0
     160     .06       0     200      .1       0
#XS Ineff= 2 , 0
                           99.83         1267.55
Permanent Ineff=
       F       F
Bank Sta=66.24,85.7
XS Rating Curve= 0 ,0
Exp/Cntr(USF)=0,0
Exp/Cntr=0.3,0.1
